--- DEVILCK.prj (project) ---

Proj Title=DEVILCK
Current Plan=p01
Default Exp/Contr=0,0
English Units
Geom File=g01
Flow File=f01
Plan File=p01
BEGIN DESCRIPTION:
END DESCRIPTION:
DSS Export Rating Curves= 0
DSS Export Rating Curve Sorted= 0
DSS Export Volume Flow Curves= 0
DXF OffsetX= 0
DXF OffsetY= 0
DXF ScaleX= 0
DXF ScaleY= 0

--- DEVILCK.p01 (plan) ---

Plan Title=Floodplain
Program Version=4.00
Geom File=g01
Flow File=f01
K Sum by GR=0
Std Step Tol=0.01
Critical Tol=0.01
Num of Std Step Trials=20
Max Error Tol=0.3
Flow Tol Ratio=0.001
Split Flow NTrial=30
Split Flow Tol=0.02
Split Flow Ratio=0.02
Log Output Level=0
Friction Slope Method=1
Unsteady Friction Slope Method=2
Unsteady Bridges Friction Slope Method=1
Global Log Level=0
CheckData=False
Run HTab=0
Run UNet=0
Run PostProcess=0
UNET Theta=0
UNET Theta Warmup=0
UNET ZTol=0
UNET ZSATol=0
UNET MxIter=0
UNET MaxInSteps=0
UNET DtIC=0
UNET DtMin=0
UNET MaxCRTS=0
UNET WFStab=0
UNET SFStab=0
UNET WFX=0
UNET SFX=0
UNET DSS MLevel=0
UNET DZMax Abort=0
UNET Convert EG Bridges=0
UNET Use Existing IB Tables=0
UNET Froude Limit=0
UNET Froude Power=0
Write IC File=0
Echo Input=False
Echo Output=False
Write Detailed=0

--- DEVILCK.f01 (steady flow) ---

Flow Title=2010 USGS WV Regression Equation
Program Version=4.00
Number of Profiles=1
Profile Names=P100yr
River Rch & RM=DEVILCK,Main      ,29586.8
537.2149
River Rch & RM=DEVILCK,Main      ,28972.1
539.3451
River Rch & RM=DEVILCK,Main      ,28186.8
597.8212
River Rch & RM=DEVILCK,Main      ,27836.8
629.9500
River Rch & RM=DEVILCK,Main      ,26054
685.8411
River Rch & RM=DEVILCK,Main      ,24520.6
830.1149
River Rch & RM=DEVILCK,Main      ,24520.6
748.5392
River Rch & RM=DEVILCK,Main      ,23420
862.6508
River Rch & RM=DEVILCK,Main      ,20836.8
927.5962
River Rch & RM=DEVILCK,Main      ,18731
1030.329
River Rch & RM=DEVILCK,Main      ,15840
1082.582
River Rch & RM=DEVILCK,Main      ,11721.1
1199.593
River Rch & RM=DEVILCK,Main      ,5995.3
1299.395
River Rch & RM=DEVILCK,Main      ,5415.4
1849.036
River Rch & RM=DEVILCK,Main      ,438.8
1943.616
River Rch & RM=DEVILCK,Main      ,438.8
1942.870
Boundary for River Rch & Prof#=DEVILCK,Main      ,1
Up Type=0
Dn Type=3
Dn Slope=0.00406

--- DEVILCK.g01 (geometry) ---

Geom Title=LiDAR
Program Version=4.10

River Reach=DEVILCK         ,Main
Reach XY= 30
     2158919.808      229079.377      2158325.19      228456.764
     2155776.796       224622.78     2155189.734        224498.9
     2154109.873      223636.052      2153910.22      223725.462
     2153605.533      223420.775     2153680.186      223198.553
     2153424.109      222654.282     2152797.373      222214.178
     2151964.301      222243.114     2151261.566      221851.548
      2151132.66      221453.761     2150188.649      221063.136
     2149643.076      220434.229     2149396.983      220642.563
     2149080.576      220438.136     2148285.004      220399.073
     2147848.806      220085.271     2147406.097      220198.552
      2146851.41      219985.011     2144919.769      219804.238
     2144364.213      219281.235      2143920.42        219123.9
     2142955.793      218132.146      2141961.87      218418.605
     2141553.884      218255.844     2141541.948      218021.469
      2140874.63      217786.009     2138365.757      218367.823

Type RM Length L Ch R = 1 ,29586.8 ,210.6,199.9,193.9
XS GIS Cut Line= 3
     2159423.783      228879.018     2158916.646       229069.89
     2158440.884      229381.533
#Sta/Elev= 30
       0 2516.29    84.9 2512.89   189.3 2510.45   199.1 2510.56   261.1 2508.78
   313.4 2508.05   365.6  2506.8  477.052506.319   496.2 2506.19   512.5 2504.83
   528.8 2504.53   534.4 2504.07   541.9 2503.69   549.4 2504.08     568 2505.56
   590.9 2505.23   597.4 2506.05     604 2507.92  615.39  2507.7   659.5 2508.99
   672.6 2508.81   698.8  2509.5   731.4 2509.69   757.6 2510.54   819.7  2511.3
   829.5 2512.01   878.5 2512.48   943.9 2514.46   963.5 2514.44  1110.6 2517.69
#Mann= 5 ,-1 , 0
       0     .12       0  477.05     .08       0   534.4    .045       0
   549.4     .08       0  615.39     .12       0
Bank Sta=534.4,549.4
XS Rating Curve= 0 ,0
Exp/Cntr=0.3,0.1

Type RM Length L Ch R = 1 ,29386.9 ,410,414.8,420.1
XS GIS Cut Line= 3
     2159148.547      228531.086     2158776.275      228930.699
     2158412.649      229337.963
#Sta/Elev= 30
       0 2545.87     9.8  2542.6    22.9 2535.05    29.4 2532.23    42.5 2530.63
   51.612531.337      85 2533.45   93.632535.876   107.9 2534.53   143.9 2527.78
     206 2517.72  268.242510.047  303.852505.859   320.5 2504.86   376.1 2504.17
   441.5 2504.78   461.1 2503.96   490.6 2504.11   510.2 2505.17  531.432503.816
  541.672502.797   549.4  2502.6     556 2502.78   565.8 2504.46   585.4 2505.68
   636.52505.554   925.4 2511.86  1000.6 2514.09  1043.1 2516.76  1092.1 2517.79
#Mann= 9 ,-1 , 0
       0     .12       0   51.61    .016       0   93.63     .12       0
  268.24    .016       0  303.85     .12       0  531.43     .08       0
  541.67    .045       0     556     .08       0   636.5     .12       0
Bank Sta=541.67,556
XS Rating Curve= 0 ,0
Exp/Cntr=0.3,0.1

Type RM Length L Ch R = 1 ,28972.1 ,432.4,435.3,437.1
XS GIS Cut Line= 3
     2158903.182      228321.521     2158473.629      228658.445
     2158028.333      228975.297
#Sta/Elev= 30
       0 2526.54    29.4 2527.73    32.7 2527.59   38.152525.916      49 2520.62
    55.6 2519.12     121 2514.76   232.1 2503.89   323.6 2501.94   356.3  2502.6
  369.412501.631   405.4 2502.73  463.352501.895   493.6 2502.57   542.6 2501.72
   549.2  2501.5  561.122501.721  590.452502.621   670.3 2505.08   758.6 2505.66
     775 2504.88   797.9 2506.29   928.8 2509.38   964.8 2508.95   974.6 2506.58
     991 2505.78   994.3    2506  1004.1  2509.4  1013.9 2510.97  1092.4 2513.44
#Mann= 7 ,-1 , 0
       0    .016       0   38.15     .12       0  369.41     .08       0
  463.35     .04       0   542.6    .045       0  561.12     .04       0
  590.45     .12       0
Bank Sta=542.6,561.12
XS Rating Curve= 0 ,0
Exp/Cntr=0.3,0.1

Type RM Length L Ch R = 1 ,28536.8 ,350.7,350,349.3
XS GIS Cut Line= 3
     2158700.485      228019.606     2158231.178      228298.653
     2157761.871        228577.7
#Sta/Elev= 30
       0 2521.18     9.8 2520.31    32.7 2515.99    42.5 2514.49    55.6 2513.02
    68.7 2512.06   137.3 2510.06   179.8 2508.34   196.2 2508.01   202.7 2506.96
   209.2 2507.46     219  2507.2   258.3  2505.7   300.8 2503.48  351.452502.335
     376 2501.19   379.3 2501.18   833.7 2501.18   879.5  2502.2   889.3 2502.83
   899.1 2502.97   908.9  2503.5   915.4 2503.41   935.1 2505.16   961.2 2506.36
   990.6 2508.72  1013.5 2509.75    1043 2510.36  1069.1 2511.49    1092 2511.99
#Mann= 4 ,-1 , 0
       0     .12       0  351.45    .016       0     376    .045       0
   833.7     .12       0
Bank Sta=376,833.7
XS Rating Curve= 0 ,0
Exp/Cntr=0.3,0.1

Type RM Length L Ch R = 1 ,28186.8 ,348.8,350,351.2
XS GIS Cut Line= 3
     2158507.252      227708.667     2158046.389       228001.45
     2157585.527      228294.233
#Sta/Elev= 30
       0 2516.28   15.912515.144    19.6 2514.69    29.4 2511.61    32.7    2511
    62.1 2508.21   127.5 2506.01   189.6 2503.18  233.622502.702   245.2 2502.35
     255 2502.43   258.3 2502.27   264.8 2501.28   268.1 2501.19   271.4 2501.18
     752 2501.19   794.5 2503.02   814.1  2503.3   820.6 2503.67   850.1 2504.41
   876.2 2505.66   908.9 2506.76   918.7 2506.48   948.1 2506.86   977.6 2507.94
   993.9    2508    1007  2508.8  1046.2 2510.53  1059.3 2512.03    1092 2513.24
#Mann= 5 ,-1 , 0
       0    .016       0   15.91     .12       0  233.62     .04       0
   268.1    .045       0     752     .12       0
Bank Sta=268.1,752
XS Rating Curve= 0 ,0
Exp/Cntr=0.3,0.1

Type RM Length L Ch R = 1 ,27836.8 ,352.5,350,347.5
XS GIS Cut Line= 3
     2158346.037       227432.35     2157869.801      227699.399
     2157393.564      227966.447
#Sta/Elev= 30
       0 2546.45     9.8 2545.13    13.1 2544.33    19.6 2541.56    26.2 2538.05
    29.4 2535.91    39.2 2528.38      49 2521.97    52.3 2520.44    62.1 2519.45
    75.2 2516.58   80.892516.098   114.4 2517.87  120.092518.836   127.5 2520.58
   130.8 2520.78   137.3 2519.47   166.7 2512.12   183.1 2508.74   232.1 2501.87
   238.7  2501.2   241.9 2501.18   840.2 2501.22   850.1 2502.39  863.442502.601
   879.5 2502.39   902.4 2503.23   954.7 2503.91  1023.3 2506.27    1092 2509.58
#Mann= 7 ,-1 , 0
       0     .12       0   80.89    .016       0  120.09     .12       0
   232.1     .04       0   238.7    .045       0   840.2     .04       0
  863.44     .12       0
Bank Sta=238.7,840.2
XS Rating Curve= 0 ,0
Exp/Cntr=0.3,0.1

Type RM Length L Ch R = 1 ,27486.8 ,574.7,575.7,576.7
XS GIS Cut Line= 3
     2158127.813      227085.761     2157683.808      227403.529
     2157239.804      227721.297
#Sta/Elev= 30
       0  2514.1    16.4 2513.04    42.5 2513.08    45.8 2513.87    52.3 2517.28
   56.322518.399    62.1 2518.89    91.5 2518.86    94.8 2518.75   98.462517.987
   101.4 2516.82   114.4  2509.3   117.7 2508.14     121 2507.48   130.8 2506.84
   147.1 2504.76   156.9 2503.95     170 2504.12   179.8 2503.42   212.5 2502.25
   222.3  2501.2   225.6 2501.18     886 2501.19   895.8 2502.28   925.3 2504.03
   938.3 2503.63   961.2 2504.44   980.8 2504.19  1033.2 2504.72    1092 2506.76
#Mann= 5 ,-1 , 0
       0     .12       0   56.32    .016       0   98.46     .12       0
   222.3    .045       0     886     .12       0
Bank Sta=222.3,886
XS Rating Curve= 0 ,0
Exp/Cntr=0.3,0.1

Type RM Length L Ch R = 1 ,26911.1 ,856.7,857.1,857.6
XS GIS Cut Line= 2
     2157910.314       226570.09     2156668.995      227377.382
#Sta/Elev= 30
       0 2538.51    52.4  2527.6    68.8 2525.07    81.9 2523.73   160.5 2517.05
   163.8  2517.3  175.68 2521.23   183.4 2521.73   206.4 2521.24   212.9 2520.63
  219.622518.346   232.6  2510.4   239.2 2507.79   245.7 2506.57  274.65 2503.73
   298.1 2501.19 1195.04 2501.18  1195.7 2501.18  1231.8 2503.54  1287.5 2505.58
  1356.2  2509.2  1382.5 2509.78  1408.7 2511.87  1428.3 2510.43  1434.9 2510.37
    1448 2512.02  1457.8 2512.65  1464.4 2511.92  1470.9 2510.13  1480.7 2510.56
#Mann= 6 ,-1 , 0
       0     .12       0  175.68    .016       0  219.62     .12       0
  274.65     .04       0   298.1    .045       0  1195.7     .12       0
Bank Sta=298.1,1195.7
XS Rating Curve= 0 ,0
Exp/Cntr=0.3,0.1

Type RM Length L Ch R = 1 ,26054   ,867.2,866,864.8
XS GIS Cut Line= 2
     2157497.988      225832.243     2156065.696       226726.34
#Sta/Elev= 30
       0 2524.54    19.7 2524.65    36.1 2527.08   63.322527.193   84.932525.819
  119.752521.769     141 2520.26   167.2 2520.02     200 2518.76   268.8 2513.97
   288.5 2513.08   337.7  2509.2  409.282502.173   419.6 2501.18  1265.5 2501.18
 1285.972502.743  1327.8 2504.95  1367.2 2506.11  1373.7 2505.75  1386.8 2503.93
  1396.7 2503.69  1409.8 2506.03    1459 2508.88  1508.1 2509.93  1537.6 2511.41
  1550.8  2511.2  1583.12512.741  1645.8 2517.03  1675.3 2520.22  1688.4 2521.09
#Mann= 9 ,-1 , 0
       0     .12       0   63.32    .016       0   84.93     .08       0
  119.75     .12       0  409.28     .04       0   419.6    .045       0
  1265.5     .04       0 1285.97     .12       0  1583.1     .06       0
Bank Sta=419.6,1265.5
XS Rating Curve= 0 ,0
Exp/Cntr=0.3,0.1

Type RM Length L Ch R = 1 ,25187.9 ,668.9,667.4,665.5
XS GIS Cut Line= 2
     2156964.133      225103.077     2155492.779      226131.722
#Sta/Elev= 30
       0 2557.71   36.942556.195    52.4 2555.57    75.4 2552.27   140.9 2542.64
   167.1 2537.19   173.6  2533.8  188.96 2521.04   193.3 2518.42   199.8 2516.65
  229.342518.104   239.2 2516.98     249 2510.74   252.3 2509.75  262.012509.201
  265.382508.892   278.5  2502.2     285 2501.19  1418.5 2501.18  1500.22503.261
 1570.852509.375 1615.812517.229  1628.2 2519.14 1653.462525.639  1677.3 2531.22
  1705.9 2532.33 1707.062532.372  1736.3 2533.26 1748.172539.545  1795.3 2547.97
#Mann= 15 ,-1 , 0
       0    .016       0   36.94     .12       0  188.96    .016       0
  229.34     .08       0  262.01     .12       0  265.38     .04       0
     285    .045       0  1418.5     .04       0  1500.2     .12       0
 1570.85    .016       0 1615.81     .12       0 1653.46     .06       0
  1705.9     .08       0 1707.06    .016       0 1748.17     .12       0
Bank Sta=285,1418.5
XS Rating Curve= 0 ,0
Exp/Cntr=0.3,0.1

Type RM Length L Ch R = 1 ,24520.6 ,421.9,411.1,400.3
XS GIS Cut Line= 2
     2156738.439      224360.889     2155366.911      225485.021
#Sta/Elev= 30
       0 2522.35    13.1 2521.72    36.1 2518.45    62.3 2517.29    91.8 2513.41
   121.3 2511.57  130.972512.029   144.2 2512.35   147.5 2511.69   154.1 2509.43
  175.152509.091   186.8 2508.72   206.5 2507.54   233.62505.167   242.6 2503.92
   252.4    2503   262.2 2501.44   268.8 2501.19  1442.3 2501.19  1458.7 2501.76
  1504.6 2502.22 1512.242502.911    1521 2504.78  1527.5 2505.42 1593.862507.027
  1684.8 2510.35 1694.992511.389 1708.022511.829  1763.5 2512.05  1773.4 2512.83
#Mann= 10 ,-1 , 0
       0     .12       0  130.97    .016       0  175.15     .12       0
   233.6     .04       0   268.8    .045       0  1442.3     .04       0
 1512.24     .06       0 1593.86     .08       0 1694.99     .12       0
 1708.02     .06       0
Bank Sta=268.8,1442.3
XS Rating Curve= 0 ,0
Exp/Cntr=0.3,0.1

Type RM Length L Ch R = 1 ,24109.5 ,121.6,120.8,120.3
XS GIS Cut Line= 3
     2156004.932      224100.472      2155497.12      225259.327
     2155310.488      225428.597
#Sta/Elev= 30
       0 2554.95   150.8 2533.66   272.1 2520.05     318 2516.74   327.8 2513.03
  333.592512.641     354  2512.8  367.012510.343   383.5 2508.46   409.7 2501.23
     413 2501.18   809.6 2501.25     826 2502.89  839.212506.558   858.8  2511.9
  871.462513.589   881.7 2515.67   921.1 2517.98   950.6 2515.32    1003 2504.34
  1016.1 2502.84 1095.722501.673 1129.44  2502.4  1163.72502.338 1293.032504.905
 1299.922505.172 1387.842509.085 1433.292510.762  1464.8 2513.48  1517.2 2513.84
#Mann= 14 ,-1 , 0
       0     .12       0  333.59    .016       0  367.01     .12       0
   409.7    .045       0   809.6     .12       0  839.21     .06       0
  871.46     .12       0 1095.72     .06       0 1129.44     .04       0
  1163.7     .06       0 1293.03     .12       0 1299.92     .06       0
 1387.84     .12       0 1433.29    .016       0
Bank Sta=409.7,809.6
XS Rating Curve= 0 ,0
Exp/Cntr=0.3,0.1

Type RM Length L Ch R = 1 ,23988.6 ,220,220.6,219.4
XS GIS Cut Line= 2
     2155879.064      224039.709     2155388.613      225272.347
#Sta/Elev= 30
       0 2559.02   219.5 2529.49   350.5 2516.42   399.6  2509.1   419.3 2508.77
   455.3  2495.8   478.2 2490.78   560.1 2489.03     570 2489.01  574.762488.976
   576.5 2488.96  609.29 2489.15  745.482490.375   763.2 2491.51  819.022501.367
   845.1 2503.35   887.7 2504.16   959.8 2500.03   989.2 2502.06  1012.2 2499.02
    1081 2499.63  1094.1 2494.38  1100.6 2495.61  1110.4 2500.31  1130.1 2500.13
 1258.842505.859  1290.6 2506.35 1319.672508.385 1324.682508.656  1326.6 2508.74
#Mann= 10 ,-1 , 0
       0     .12       0   560.1    .045       0     570     .12       0
  574.76     .06       0  609.29     .12       0  745.48     .06       0
  819.02     .12       0 1258.84    .016       0 1319.67     .12       0
 1324.68    .016       0
#XS Ineff= 2 , 0
                           621.1         2491.02
Permanent Ineff=
       F       F
Bank Sta=560.1,570
XS Rating Curve= 0 ,0
Exp/Cntr=0.3,0.1

Type RM Length L Ch R = 1 ,23768   ,343.3,348,347.1
XS GIS Cut Line= 2
     2155706.104       223959.63     2155242.562      225103.728
#Sta/Elev= 30
       0 2546.21    19.6 2543.26   101.5 2533.62   153.9 2528.77   229.2 2519.97
   301.2 2513.42   458.4 2495.32   474.8    2492   497.7 2490.71   527.2 2484.32
   530.4 2483.01     537 2477.91   543.5 2476.97   551.7 2477.95   559.9 2479.57
     573 2479.35   602.5 2480.76   615.6 2479.75   651.6 2481.74     668 2481.75
   690.9 2485.67   700.7 2486.51   792.4 2488.93   867.7 2492.57  978.822494.646
 1110.682501.148  1129.7 2503.09  1159.1 2503.65    1182 2508.41  1234.4 2512.14
#Mann= 5 ,-1 , 0
       0     .12       0     537    .045       0   551.7     .12       0
  978.82    .016       0 1110.68     .12       0
Bank Sta=537,551.7
XS Rating Curve= 0 ,0
Exp/Cntr=0.3,0.1

Type RM Length L Ch R = 1 ,23420   ,480.7,483.1,480
XS GIS Cut Line= 2
     2155496.034      223869.353     2154982.146      224902.339
#Sta/Elev= 30
       0 2532.09     9.8 2528.79    91.8 2519.82     213 2503.39   321.2 2494.26
   340.9 2491.47   367.1 2491.07   485.1 2479.81     531 2477.86   557.2 2478.35
   612.9 2475.16   629.3 2476.44   645.7 2474.86   671.9 2476.33  689.43 2474.75
   694.9 2473.36   704.7 2474.86   711.3 2479.57   714.5 2480.47   737.5 2482.39
     767 2491.24   783.4 2493.64   809.6 2493.26  843.882487.209  860.562486.534
   904.6 2488.63   976.8 2499.22  1084.9 2528.68  1114.4 2534.75  1153.8 2540.22
#Mann= 5 ,-1 , 0
       0     .12       0  689.43    .045       0   704.7     .12       0
  843.88    .016       0  860.56     .12       0
Bank Sta=689.43,704.7
XS Rating Curve= 0 ,0
Exp/Cntr=0.3,0.1

Type RM Length L Ch R = 1 ,22936.8 ,342.6,350,351.4
XS GIS Cut Line= 3
     2155156.991      223702.175     2154931.766      224274.496
     2154676.421      224747.029
#Sta/Elev= 30
       0 2503.82     9.8 2503.97   101.4  2489.1   206.1 2480.59     265 2479.15
   356.6  2479.8   451.5 2478.03   520.2 2478.08   539.8 2477.07   556.2 2474.14
  573.182474.023   598.7 2474.33  609.052471.722   618.3  2470.2   624.9 2471.74
   654.3 2476.31  688.232475.774     733 2476.85   762.4 2478.71   775.5 2481.12
   791.9 2486.43     805 2488.73   837.8  2503.7   883.6 2521.81   922.9 2531.96
   945.8 2534.98  1001.5 2537.88  1037.5 2537.25  1096.5 2527.83  1152.2 2520.95
#Mann= 5 ,-1 , 0
       0     .12       0  573.18     .08       0  609.05    .045       0
   624.9     .08       0  688.23     .12       0
#XS Ineff= 2 , 0
                           656.5         2477.32
Permanent Ineff=
       F       F
Bank Sta=609.05,624.9
XS Rating Curve= 0 ,0
Exp/Cntr=0.3,0.1

Type RM Length L Ch R = 1 ,22586.8 ,233.4,232.8,229.9
XS GIS Cut Line= 3
     2155001.876      223581.608      2154712.03      224041.972
     2154396.958      224502.946
#Sta/Elev= 30
       0  2514.6    65.5 2498.04    78.6 2493.26   173.7 2479.54   245.8 2477.71
   409.6 2477.48   452.2  2475.2   468.6 2471.89  479.342472.309   501.4 2471.52
   530.9 2473.01   536.5 2471.07   540.7 2469.52   550.5 2471.24   563.6 2473.25
  603.052472.319   697.5 2475.92   707.3 2481.37   723.6 2483.88   756.2 2497.89
     766 2500.37   795.4  2503.2   824.8 2499.43   870.5 2489.52   916.2 2487.41
   929.3 2495.92     975 2494.59   988.1 2495.62  1056.7 2510.52  1102.4 2522.29
#Mann= 5 ,-1 , 0
       0     .12       0  479.34     .08       0   536.5    .045       0
   550.5     .08       0  603.05     .12       0
Bank Sta=536.5,550.5
XS Rating Curve= 0 ,0
Exp/Cntr=0.3,0.1

Type RM Length L Ch R = 1 ,22354   ,458.1,467.2,444.5
XS GIS Cut Line= 2
     2154792.909      223478.728     2154225.201        224419.7
#Sta/Elev= 30
       0 2503.27    39.4 2494.48    72.2 2489.33   108.3 2484.36   177.2 2477.91
   213.2 2475.85   416.6 2474.22   436.3 2473.02     456 2469.93  481.212470.637
   492.1  2469.4   501.9  2468.4  506.182469.388   518.3 2472.54   551.1 2470.94
  602.992473.228   636.4 2473.55  668.762477.973   695.5 2478.87   708.6 2481.84
  734.542484.072  754.41 2484.83   793.9  2486.2  822.572484.687   849.6 2487.18
   898.8 2500.56   941.5 2508.95  1020.2 2518.49  1049.8 2523.58    1099 2534.68
#Mann= 9 ,-1 , 0
       0     .12       0  481.21     .08       0   492.1    .045       0
  506.18     .08       0  602.99     .12       0  668.76     .06       0
  734.54     .12       0  754.41     .06       0  822.57     .12       0
#XS Ineff= 2 , 0
                          605.64         2474.58
Permanent Ineff=
       F       F
Bank Sta=492.1,506.18
XS Rating Curve= 0 ,0
Exp/Cntr=0.3,0.1

Type RM Length L Ch R = 1 ,21886.8 ,529.7,531.1,524.3
XS GIS Cut Line= 3
     2154555.828       223316.65       2154273.4      223818.734
     2153957.392      224302.247
#Sta/Elev= 30
       0 2522.23   117.8 2498.12   127.6 2498.19   189.8 2485.82   258.6 2475.44
   301.1 2472.21   333.9 2473.63   500.8 2472.99   513.9 2469.69  537.832469.329
   556.4 2470.12   566.2 2468.53   572.8 2466.95   579.3 2468.66   589.1 2470.25
   605.4 2469.54  664.522472.522   765.3 2475.39   794.7 2478.08   817.6 2485.03
   827.4 2489.32   837.1 2490.24   856.7  2499.8   931.8 2522.61  1016.6    2541
  1042.7 2544.71  1072.1    2547  1091.7 2546.06  1130.8 2541.21  1153.7 2540.26
#Mann= 5 ,-1 , 0
       0     .12       0  537.83     .08       0   566.2    .045       0
   579.3     .08       0  664.52     .12       0
Bank Sta=566.2,579.3
XS Rating Curve= 0 ,0
Exp/Cntr=0.3,0.1

Type RM Length L Ch R = 1 ,21355.8 ,181.9,168.9,170.8
XS GIS Cut Line= 2
     2154371.034      223202.686     2153584.576        224107.2
#Sta/Elev= 30
       0 2516.98   255.4  2499.2   265.3 2499.72   324.2 2497.02   376.6 2493.59
     465 2473.36   501.1 2470.96   510.9 2469.12   527.3 2471.04  628.392469.559
   671.4    2468   687.7 2464.55   694.3 2464.08  702.092464.546   707.4 2467.49
   720.5 2469.34   733.6 2474.29   756.5 2474.97  764.992476.523   779.4 2480.25
   825.3 2482.58   864.6 2490.91   907.1 2501.87   956.3 2510.57   982.5 2514.07
  1011.9 2516.38  1064.3 2519.04  1116.7 2525.35  1149.5  2531.6  1198.6 2545.58
#Mann= 5 ,-1 , 0
       0     .12       0  628.39     .08       0   687.7    .045       0
  702.09     .08       0  764.99     .12       0
#XS Ineff= 2 , 0
          562.23 2474.19
Permanent Ineff=
       F       F
Bank Sta=687.7,702.09
XS Rating Curve= 0 ,0
Exp/Cntr=0.3,0.1

Type RM Length L Ch R = 1 ,21186.8 ,327.5,350,359.6
XS GIS Cut Line= 3
     2154242.989      223108.605      2153831.94      223593.917
     2153410.775      223945.558
#Sta/Elev= 30
       0 2516.76     141 2504.48   170.5  2503.2     200 2498.92   222.9 2497.95
   354.1 2485.58   363.9 2485.62   432.7 2478.15   488.5  2478.8  550.532475.018
   586.8 2466.93   609.8 2467.19   628.5 2465.45     636 2464.09   643.5 2465.41
  677.632469.462   704.6 2469.81     747 2472.83   760.1 2472.59   786.2 2476.61
   841.7 2490.17   871.1 2494.82   929.9 2498.86   965.8 2498.98   978.9 2498.05
  1001.8  2502.1  1050.8 2507.32  1076.9 2513.21  1148.7 2538.97  1184.7 2549.83
#Mann= 5 ,-1 , 0
       0     .12       0  550.53     .08       0   628.5    .045       0
   643.5     .08       0  677.63     .12       0
Bank Sta=628.5,643.5
XS Rating Curve= 0 ,0
Exp/Cntr=0.3,0.1

Type RM Length L Ch R = 1 ,20836.8 ,366.6,370.9,353.8
XS GIS Cut Line= 3
     2154186.676      223050.249     2153602.492      223409.044
     2153097.807       223539.89
#Sta/Elev= 30
       0 2521.96      59 2522.57   209.9 2510.88   239.5 2505.24   259.1 2504.45
   308.3 2495.48   334.6 2489.44   354.3 2482.55   423.2 2476.89   482.2 2474.15
   521.6 2469.35  563.142466.883   600.3 2465.06   662.6 2466.68     679 2464.59
   685.6 2462.82   692.1 2464.59   695.4 2466.22  723.462469.115   767.6 2472.86
   790.5 2479.75   803.6 2480.68     879 2516.23   931.5 2538.17   980.7  2555.3
    1043 2572.01  1072.5 2576.15  1111.8  2576.6  1154.5 2570.56  1206.9 2558.22
#Mann= 5 ,-1 , 0
       0     .12       0  563.14     .08       0     679    .045       0
   692.1     .08       0  723.46     .12       0
Bank Sta=679,692.1
XS Rating Curve= 0 ,0
Exp/Cntr=0.3,0.1

Type RM Length L Ch R = 1 ,20465.9 ,332,329.1,321.9
XS GIS Cut Line= 2
     2154167.909      222944.005     2153074.159      223341.575
#Sta/Elev= 30
       0  2533.9    39.3 2533.84   114.7 2527.07     259 2505.99     295 2498.25
   357.3 2478.32   370.4 2477.64     413 2469.15     495 2466.89   527.8 2467.77
   550.7  2465.5  589.352464.662   596.6 2462.83   603.2 2464.67   652.4 2462.51
     672  2465.6  705.822467.979  762.652468.681   809.7 2469.75   849.1 2473.75
   878.6 2487.39   888.4 2488.18   898.2 2495.15   957.2 2519.67  1003.1 2534.47
  1022.8  2538.5  1039.2 2539.52  1062.1 2537.68  1114.6 2525.29  1163.8 2517.62
#Mann= 5 ,-1 , 0
       0     .12       0  589.35    .045       0   603.2     .12       0
  705.82     .08       0  762.65     .12       0
#XS Ineff= 2 , 0
          522.25 2468.77  710.23         2468.88
Permanent Ineff=
       F       F
Bank Sta=589.35,603.2
XS Rating Curve= 0 ,0
Exp/Cntr=0.3,0.1

Type RM Length L Ch R = 1 ,20136.8 ,317.9,315.5,308.6
XS GIS Cut Line= 3
     2154052.241      222623.684     2153599.523      222904.679
     2153043.419      223180.188
#Sta/Elev= 30
       0 2594.48    75.2 2576.45     170 2555.87   228.8 2537.38   300.7    2520
   326.9 2512.75   405.4 2488.77   444.6 2475.52   464.2 2472.65   496.9 2463.02
  513.482463.451  524.412462.908   532.8 2461.14   540.3  2462.9   578.6 2464.62
   601.4 2463.26  633.28 2464.56     670 2468.13   732.1 2467.15   771.3 2469.29
   823.5 2481.39   898.7 2488.81   921.5  2492.4   937.9  2496.8   950.9 2496.92
   960.7 2499.91  1003.2 2500.85  1081.6 2498.32  1101.2 2496.83  1153.4 2499.75
#Mann= 5 ,-1 , 0
       0     .12       0  513.48     .07       0  524.41    .045       0
   540.3     .07       0  633.28     .12       0
Bank Sta=524.41,540.3
XS Rating Curve= 0 ,0
Exp/Cntr=0.3,0.1

Type RM Length L Ch R = 1 ,19821.3 ,390.7,384.5,377
XS GIS Cut Line= 2
     2153839.784      222360.672     2152930.062      223093.311
#Sta/Elev= 30
       0 2592.98    94.9 2562.93   160.3  2545.1     193 2534.74   258.5 2519.89
   327.2 2501.61   418.8 2482.81   464.6 2473.92   474.4 2472.81   487.5    2467
   497.3 2461.09   500.6 2459.98   507.1 2459.58  512.782461.112     517 2462.22
     530 2463.14  567.11 2462.84  577.892463.295   664.2 2466.54   683.8 2470.88
   723.1 2476.48   752.5 2479.17   801.6 2482.11   860.5 2483.43   912.8 2485.67
   968.5 2486.31  1050.3 2491.63  1099.4 2493.61  1151.7 2491.59  1168.1 2493.39
#Mann= 5 ,-1 , 0
       0     .12       0   497.3    .045       0  512.78     .12       0
  567.11     .06       0  577.89     .12       0
#XS Ineff= 2 , 0
                           629.1         2471.08
Permanent Ineff=
       F       F
Bank Sta=497.3,512.78
XS Rating Curve= 0 ,0
Exp/Cntr=0.3,0.1

Type RM Length L Ch R = 1 ,19436.8 ,265.8,260.8,254.6
XS GIS Cut Line= 3
     2153433.051      222078.802     2153119.175      222537.607
     2152791.256      222976.485
#Sta/Elev= 30
       0 2535.93    98.1  2518.6   294.3 2491.05   346.6 2482.13   398.9 2475.88
   503.6 2465.92   548.4 2459.56   552.6 2459.07   563.4 2459.66   585.4 2464.37
   608.4 2464.55   621.5 2467.33   644.5    2470     779 2476.96   828.2 2477.94
   900.4 2481.72   936.4 2481.72     966 2483.09   972.5 2482.65   979.1 2480.09
   992.2  2479.7  1005.3  2482.5  1011.9  2482.5  1021.7 2480.56  1031.6 2482.92
  1034.9 2485.68    1048 2500.55  1057.8 2507.39  1070.9 2512.16  1103.8 2520.82
#Mann= 3 ,-1 , 0
       0     .12       0   548.4    .045       0   563.4     .12       0
Bank Sta=548.4,563.4
XS Rating Curve= 0 ,0
Exp/Cntr=0.3,0.1

Type RM Length L Ch R = 1 ,19176   ,450.8,445,436.3
XS GIS Cut Line= 2
     2153131.451      221872.825     2152700.896        222919.7
#Sta/Elev= 30
       0 2569.36     9.8 2566.73    65.4 2545.88    94.9 2536.34   160.3 2521.41
   196.3 2511.54   235.6 2499.02   287.9 2485.76   333.7 2475.56   363.1  2470.5
   402.4 2467.26     530 2461.82   552.9 2461.65   566.1 2458.68   572.5 2457.36
   581.1  2458.8   592.2 2460.21     615 2459.01   641.2 2462.01   700.1 2464.73
   729.6 2467.13     880  2472.2   922.6 2475.47   935.7 2474.88   974.9 2476.42
   994.6 2473.46  1004.4 2476.63  1030.5 2495.36  1040.4 2500.43    1132 2532.76
#Mann= 3 ,-1 , 0
       0     .12       0   566.1    .045       0   581.1     .12       0
#XS Ineff= 2 , 0
          551.83 2463.67
Permanent Ineff=
       F       F
Bank Sta=566.1,581.1
XS Rating Curve= 0 ,0
Exp/Cntr=0.3,0.1

Type RM Length L Ch R = 1 ,18731   ,342.1,344.2,347.7
XS GIS Cut Line= 2
     2152681.798      221733.936     2152589.784      222853.728
#Sta/Elev= 30
       0 2561.79    65.5 2544.53   127.8 2531.96     154  2525.3   252.2 2496.92
   314.5  2484.6   330.8 2479.21   340.7 2478.33   353.8 2474.24     380 2470.32
   393.1 2469.72   402.9 2467.48   432.4 2468.04   448.8 2464.33   471.7 2463.04
   491.4 2456.22   524.1 2454.55   532.2 2452.88   540.5 2452.27   547.2    2453
   576.5 2458.17   635.5  2458.6   818.9 2466.68   871.3 2467.39   907.4 2469.64
   923.8 2472.94   933.6 2473.26  1015.5 2505.95  1041.7 2514.18  1123.6 2536.06
#Mann= 3 ,-1 , 0
       0     .12       0   532.2    .045       0   547.2     .12       0
#XS Ineff= 2 , 0
          498.57 2459.52
Permanent Ineff=
       F       F
Bank Sta=532.2,547.2
XS Rating Curve= 0 ,0
Exp/Cntr=0.3,0.1

Type RM Length L Ch R = 1 ,18386.8 ,344.4,351.1,354
XS GIS Cut Line= 3
     2152400.484      221709.036     2152315.083      222247.411
     2152186.914      222788.782
#Sta/Elev= 30
       0 2529.84    35.9 2530.15   107.7 2528.47   264.4 2507.82   326.4 2498.08
   372.1 2488.71   385.2 2485.55   430.9 2470.41   443.9 2464.78   450.4 2464.99
   460.2 2461.58   486.4 2458.12   502.7  2453.8   525.5 2453.34   537.6 2448.97
   548.4 2448.66   552.6 2448.93   597.5  2453.4   643.3 2453.05   662.9 2451.94
   695.6 2454.05   767.6 2456.35   797.1 2460.04     820 2465.09   829.8 2465.69
   849.4 2472.27     892 2484.42   990.2  2511.1  1022.9 2518.45  1101.4 2549.41
#Mann= 3 ,-1 , 0
       0     .12       0   537.6    .045       0   552.6     .12       0
Bank Sta=537.6,552.6
XS Rating Curve= 0 ,0
Exp/Cntr=0.3,0.1

Type RM Length L Ch R = 1 ,18035.7 ,261.8,269.5,272.4
XS GIS Cut Line= 3
     2152225.069      221686.968     2151969.369       222240.26
     2151781.109      222740.455
#Sta/Elev= 30
       0 2555.76    72.1 2533.62   134.4 2521.13     249 2494.77   281.8 2484.08
   304.8 2474.73   327.7 2463.42   363.8 2452.63   406.4 2448.06   455.5 2448.29
   498.1 2446.01     521 2447.54   573.5 2447.68  600.042445.652  603.982444.678
   616.1  2444.3  619.972444.681   632.5 2449.38  665.362449.841   714.4 2451.64
   740.7 2462.82   750.5  2464.7   766.9 2472.74   793.1 2482.81   835.8 2494.13
   871.8 2497.41   983.3 2499.83  1016.1 2496.34  1055.4 2507.76    1144 2520.45
#Mann= 5 ,-1 , 0
       0     .12       0  600.04     .08       0  603.98    .045       0
  619.97     .08       0  665.36     .12       0
#XS Ineff= 2 , 0
          424.35 2449.79
Permanent Ineff=
       F       F
Bank Sta=603.98,619.97
XS Rating Curve= 0 ,0
Exp/Cntr=0.3,0.1

Type RM Length L Ch R = 1 ,17766.3 ,538.3,545.3,540.9
XS GIS Cut Line= 2
     2152046.382      221596.783     2151482.146      222593.311
#Sta/Elev= 30
       0 2518.98    32.7 2510.69     193 2479.09   271.6 2466.12   310.8 2454.87
     373 2450.26   418.8 2444.34   441.7 2444.85   454.8 2442.66   484.2  2444.7
   503.9 2444.99  523.582443.971  537.452442.883   546.4 2441.98     553 2442.92
   592.2 2445.56   664.2 2444.32   683.8 2452.08   693.6 2452.55   696.9 2453.66
   706.7 2461.19   710.8 2462.54   723.1 2466.55   775.4 2478.51   824.5 2493.61
     854 2501.54   909.6 2512.43   942.3 2521.35  1056.8 2562.88  1145.2 2598.57
#Mann= 5 ,-1 , 0
       0     .12       0  523.58     .08       0  537.45    .045       0
     553     .08       0   710.8     .12       0
#XS Ineff= 2 , 0
                           622.3         2448.33
Permanent Ineff=
       F       F
Bank Sta=537.45,553
XS Rating Curve= 0 ,0
Exp/Cntr=0.3,0.1

Type RM Length L Ch R = 1 ,17221   ,204.3,207.4,210.1
XS GIS Cut Line= 2
     2151798.118      221456.158     2151107.146      222351.992
#Sta/Elev= 30
       0 2571.26    29.5 2564.48    65.6 2553.73    98.4 2546.42   131.2 2535.47
     164 2523.36   236.1 2492.61   298.4 2463.46   347.6 2448.82   360.7 2447.76
   377.1    2444   475.5 2443.06   524.7    2439   544.4 2440.52   560.8 2438.75
   580.4 2440.53   593.6 2437.26   596.8 2436.97     610 2437.36   619.8 2439.09
   636.2 2448.33     646 2449.96   662.4 2460.93   695.2 2477.92   764.1 2511.16
   849.3 2550.04   875.6 2564.29   983.8 2616.78  1101.8 2668.06  1131.4 2679.32
#Mann= 3 ,-1 , 0
       0     .12       0   593.6    .045       0     610     .12       0
#XS Ineff= 2 , 0
          540.21  2445.2
Permanent Ineff=
       F       F
Bank Sta=593.6,610
XS Rating Curve= 0 ,0
Exp/Cntr=0.3,0.1

Type RM Length L Ch R = 1 ,17013.6 ,462.6,459.3,451.3
XS GIS Cut Line= 3
     2151725.056      221395.087     2151260.264      221825.718
      2150877.15      222202.399
#Sta/Elev= 30
       0 2562.19    91.4 2537.75   133.9 2525.12   186.2 2508.17   228.6 2492.39
   251.5 2485.77   365.8 2465.63   431.1 2452.27   499.7  2441.3   522.6 2440.01
   535.6 2440.92   555.2 2435.26   584.6 2438.77   607.5 2435.89   636.9 2438.41
   643.4  2436.6     650 2435.03  658.792436.612   679.5 2451.63   692.6 2455.42
   705.7 2464.56   748.3 2484.41   797.4 2509.41   836.7 2525.69   856.4 2532.49
   928.5 2554.54  1016.9  2576.7  1056.2 2584.39  1111.9 2597.32  1170.9 2607.49
#Mann= 3 ,-1 , 0
       0     .12       0   643.4    .045       0  658.79     .12       0
#XS Ineff= 2 , 0
          533.97 2443.48
Permanent Ineff=
       F       F
Bank Sta=643.4,658.79
XS Rating Curve= 0 ,0
Exp/Cntr=0.3,0.1

Type RM Length L Ch R = 1 ,16554.3 ,279,277.7,275
XS GIS Cut Line= 2
     2151466.521      221074.214     2150706.104      221944.005
#Sta/Elev= 30
       0 2627.69    29.5 2617.09    98.2 2598.44   130.9 2586.31   176.7 2567.45
   229.1 2539.46     288 2512.11   392.7 2470.52  468.662444.856   487.7 2440.38
   498.2 2432.94   507.3 2431.67   513.2 2432.74   523.7 2434.79  554.252435.318
   605.5 2434.97   638.2 2436.74   664.4 2448.33   674.2 2450.54   690.6 2452.05
   700.4 2454.89   762.6  2464.4   837.8 2478.99   939.3 2490.21   991.7  2499.7
    1031 2503.43  1060.4 2509.17  1076.8 2510.85  1125.9 2522.62  1155.3 2532.17
#Mann= 5 ,-1 , 0
       0     .12       0  468.66     .08       0   498.2    .045       0
   513.2     .08       0  554.25     .12       0
Bank Sta=498.2,513.2
XS Rating Curve= 0 ,0
Exp/Cntr=0.3,0.1

Type RM Length L Ch R = 1 ,16276.6 ,436.9,436.6,434.2
XS GIS Cut Line= 3
     2151230.852      220909.578      2150871.47      221398.992
     2150559.816      221833.905
#Sta/Elev= 30
       0 2617.61    32.6 2614.64    94.7 2614.45   140.4 2611.53     173 2605.64
   228.5 2587.42   267.7 2570.01   349.3  2526.8   411.3  2490.5   473.4 2449.92
   486.4 2444.84   499.5 2432.93     506 2430.98   526.62432.394   599.7  2430.3
   610.4  2429.4   614.7 2430.41  616.362430.915   623.5 2432.92   665.9 2432.48
   685.5 2441.81   705.1 2456.78   760.5 2491.46   783.4 2502.74   802.9 2508.74
   835.6 2512.84   907.3 2508.31   956.3 2511.36    1028 2525.13  1142.2 2558.08
#Mann= 5 ,-1 , 0
       0     .12       0   526.6     .08       0   599.7    .045       0
   614.7     .08       0  616.36     .12       0
Bank Sta=599.7,614.7
XS Rating Curve= 0 ,0
Exp/Cntr=0.3,0.1

Type RM Length L Ch R = 1 ,15840   ,266,265.2,264.2
XS GIS Cut Line= 2
     2150860.618      220759.978     2150292.909      221699.214
#Sta/Elev= 30
       0 2538.47    32.8 2543.53    85.2  2554.5   111.4 2557.65   157.2 2556.44
   206.4 2548.36   252.3 2533.88   278.5 2523.84   304.7 2511.71   429.2 2446.56
   442.3  2435.3  445.07 2434.01   461.9 2429.16   494.7 2430.27   524.2 2426.97
   530.7 2425.91  538.742426.969   547.1 2429.22   583.1 2429.29  635.322426.399
   671.6 2433.55   694.5 2451.55   737.1 2473.99     760 2485.32   792.8 2496.01
   832.1 2506.21   923.8 2526.26  1015.6 2548.57  1048.3 2555.44  1097.5 2562.37
#Mann= 5 ,-1 , 0
       0     .12       0  445.07     .08       0   524.2    .045       0
  538.74     .08       0  635.32     .12       0
#XS Ineff= 2 , 0
          491.66  2432.6
Permanent Ineff=
       F       F
Bank Sta=524.2,538.74
XS Rating Curve= 0 ,0
Exp/Cntr=0.3,0.1

Type RM Length L Ch R = 1 ,15574.9 ,345.5,353.8,361.1
XS GIS Cut Line= 3
     2150613.302      220635.976     2150344.267      221128.253
      2150080.09      221604.155
#Sta/Elev= 30
       0 2532.25      59 2507.36    78.7 2501.64   114.8 2495.36   183.7 2486.78
   236.2 2478.48   347.8 2466.33   505.2 2444.93   515.1 2442.64   521.6  2439.9
   524.9 2437.35   534.8 2426.06     538 2423.72   544.6 2423.49   557.7 2425.59
  562.262424.664   570.8 2422.96   577.4 2424.62     584  2425.9   610.2 2425.62
   646.2 2429.87   698.7 2452.73   767.6 2477.33     843 2508.47   859.4    2514
     902 2526.75  1013.5  2555.4  1036.4 2560.04  1075.8 2565.52  1105.3 2570.82
#Mann= 3 ,-1 , 0
       0     .12       0  562.26    .045       0   577.4     .12       0
Bank Sta=562.26,577.4
XS Rating Curve= 0 ,0
Exp/Cntr=0.3,0.1

Type RM Length L Ch R = 1 ,15221.1 ,212,208.1,202.9
XS GIS Cut Line= 3
     2150529.748      220563.467     2150112.842      220909.318
     2149671.127      221268.938
#Sta/Elev= 30
       0 2530.03    39.2 2522.98    91.4 2510.56   104.4 2505.48   117.5 2504.16
   159.9 2490.29   221.9 2473.82   267.6 2468.22   339.4 2454.12   443.8 2439.72
   453.6 2435.99   469.9  2424.8     483 2420.62   525.4 2421.32   535.2 2418.82
   541.7 2417.68   551.5 2418.78   574.4 2422.61   590.8 2421.93   626.8 2425.77
   695.5 2434.87   754.5 2455.35   764.3 2456.69   780.6 2463.66   819.9 2476.32
   901.8 2497.85   970.5 2520.41  1013.1 2529.79  1068.7 2551.75  1111.3 2566.24
#Mann= 3 ,-1 , 0
       0     .12       0   535.2    .045       0   551.5     .12       0
#XS Ineff= 2 , 0
                          577.16         2424.49
Permanent Ineff=
       F       F
Bank Sta=535.2,551.5
XS Rating Curve= 0 ,0
Exp/Cntr=0.3,0.1

Type RM Length L Ch R = 1 ,15013   ,229.7,228,227.1
XS GIS Cut Line= 2
     2150329.368      220348.519      2149614.09      221207.894
#Sta/Elev= 30
       0  2574.8    88.5 2544.84   144.3 2520.82     200 2501.03   242.6 2488.78
     318 2459.16   377.1 2444.06   390.2 2438.39   406.6 2435.99   416.4 2431.65
   439.4 2425.53  471.122421.759   501.7 2419.96  509.882415.872   514.8 2414.97
   524.6  2415.9   534.5 2418.73   588.12418.624   632.8 2417.85   668.9 2420.38
   698.4 2424.19   731.2 2434.32     741 2435.78   757.4 2443.42   813.2 2464.17
   931.2 2500.57   996.8 2526.97  1032.8 2539.54  1085.3 2556.87  1118.1  2563.4
#Mann= 5 ,-1 , 0
       0     .12       0  471.12     .08       0  509.88    .045       0
   524.6     .08       0   588.1     .12       0
#XS Ineff= 2 , 0
                          623.03         2421.27
Permanent Ineff=
       F       F
Bank Sta=509.88,524.6
XS Rating Curve= 0 ,0
Exp/Cntr=0.3,0.1

Type RM Length L Ch R = 1 ,14785   ,627.5,613.9,599.9
XS GIS Cut Line= 3
     2150162.701      220194.005     2149714.784      220779.075
     2149593.257      221195.742
#Sta/Elev= 30
       0 2607.01    29.5 2599.33    55.7  2590.6   114.6 2566.96   144.1 2553.79
   252.2 2501.96   327.5 2461.16     393 2427.39   412.6 2420.44   435.6  2417.5
  454.382416.502   481.4 2414.95   586.2 2414.11   615.7 2411.29   625.5 2410.34
     632 2411.08   638.6 2415.48   645.2 2417.34   668.1 2418.62   681.2 2418.07
  701.382420.041   730.3 2421.47   749.9  2425.4   808.6 2448.39   854.3 2462.02
   913.1 2484.34   981.6  2505.9  1020.8 2520.35  1128.4 2550.44  1170.9 2560.43
#Mann= 5 ,-1 , 0
       0     .12       0  454.38     .08       0   615.7    .045       0
     632     .08       0  701.38     .12       0
#XS Ineff= 2 , 0
          510.53  2417.1
Permanent Ineff=
       F       F
Bank Sta=615.7,632
XS Rating Curve= 0 ,0
Exp/Cntr=0.3,0.1

Type RM Length L Ch R = 1 ,14171.1 ,342.4,350,355.7
XS GIS Cut Line= 3
     2149378.673      219954.174      2149500.48      220616.525
     2149491.008      221158.794
#Sta/Elev= 30
       0 2518.36    71.9 2503.73   140.6 2484.45   176.5 2472.58   232.1 2457.94
   245.2 2452.65   261.5 2451.26   281.2 2446.11   330.2    2440   362.9 2433.97
   483.8 2422.95     510  2418.3   523.1 2409.98   529.6 2407.92   588.5 2404.88
   614.6 2407.45   634.2 2405.94   647.3 2407.35   663.6  2405.1   673.5 2403.94
     680  2405.2   696.3 2409.06   755.1 2416.22   771.5 2416.04   781.3 2419.27
   849.9 2431.98   934.8  2450.5  1062.2 2500.62  1134.1 2522.82  1215.8 2544.05
#Mann= 3 ,-1 , 0
       0     .12       0   663.6    .045       0     680     .12       0
Bank Sta=663.6,680
XS Rating Curve= 0 ,0
Exp/Cntr=0.3,0.1

Type RM Length L Ch R = 1 ,13821.1 ,354.7,350,340.8
XS GIS Cut Line= 3
     2149296.453      219943.779     2149216.991      220500.358
     2149040.493      221070.314
#Sta/Elev= 30
       0 2550.47    68.6 2550.65   104.6 2546.33   137.3 2539.53   166.7 2530.36
   212.5 2510.82   290.9 2468.52   330.1 2443.49     340 2441.55   362.8 2429.17
   382.4 2423.64   444.6 2412.79   477.2  2403.5  507.162401.794   536.1 2402.07
   554.7 2399.34   562.2  2398.6   569.7 2399.25   592.8 2402.32     618 2401.56
   716.3 2405.49   732.7 2404.75   821.2 2412.13     854 2426.02   945.8 2476.23
   958.9 2480.26   968.7  2486.1  1040.9 2518.52  1093.3 2538.02  1158.9 2558.45
#Mann= 5 ,-1 , 0
       0     .12       0  507.16     .07       0   554.7    .045       0
   569.7     .07       0   592.8     .12       0
#XS Ineff= 2 , 0
                           675.1         2406.79
Permanent Ineff=
       F       F
Bank Sta=554.7,569.7
XS Rating Curve= 0 ,0
Exp/Cntr=0.3,0.1

Type RM Length L Ch R = 1 ,13471.1 ,340.8,350,351.6
XS GIS Cut Line= 3
     2148877.751      219922.695     2148928.699       220525.91
     2148955.036      221062.898
#Sta/Elev= 30
       0 2566.38    26.2 2558.07    78.5  2533.8   127.6 2515.82   271.6 2453.02
   297.8  2443.7   363.2 2427.38     373 2426.79   405.8 2417.36   458.1 2407.16
   484.3 2396.37   520.3 2396.98   530.1 2395.18   582.5 2396.71   597.9 2394.67
   605.4 2393.97   612.9 2394.58   628.3 2398.23   670.9 2398.34     684 2396.26
   736.5 2396.77   772.6 2405.93     789  2412.3   805.3 2420.78   815.2 2423.63
   867.6 2448.97   959.4 2489.55  1067.6 2542.84  1106.9 2557.46    1143 2567.59
#Mann= 3 ,-1 , 0
       0     .12       0   597.9    .045       0   612.9     .12       0
Bank Sta=597.9,612.9
XS Rating Curve= 0 ,0
Exp/Cntr=0.3,0.1

Type RM Length L Ch R = 1 ,13121.1 ,348.8,350,350.5
XS GIS Cut Line= 3
     2148801.121      219919.867     2148660.122      220527.061
     2148576.016      221052.725
#Sta/Elev= 30
       0  2549.5      59 2522.44   124.7 2501.45   200.1 2472.34   288.7 2440.01
   367.4 2423.29   383.8 2417.85     397 2417.19     456 2402.17   498.7 2395.55
   515.1 2393.55   541.3 2393.62   551.2 2391.23   600.4 2392.99   613.5 2390.59
   620.1 2389.89  628.012390.523   636.4 2392.64     656 2393.41   685.4 2393.43
   698.5  2391.7     705 2392.94   711.5 2396.58   731.1  2413.8   740.9 2420.75
     852 2473.55   979.3 2546.02  1077.3 2591.59  1103.4 2601.39  1155.7 2616.89
#Mann= 3 ,-1 , 0
       0     .12       0   613.5    .045       0  628.01     .12       0
Bank Sta=613.5,628.01
XS Rating Curve= 0 ,0
Exp/Cntr=0.3,0.1

Type RM Length L Ch R = 1 ,12771.1 ,338.9,350,357.1
XS GIS Cut Line= 3
      2148605.32      219872.485     2148426.941      220441.102
     2148267.719       220954.15
#Sta/Elev= 30
       0 2515.14    29.5 2510.27   104.8 2491.35   268.5 2443.54   376.6  2418.9
   402.8 2410.46   435.5 2394.52   448.6 2393.99     465 2389.62   514.1 2388.52
   530.4    2386   569.7 2388.91   589.4  2385.5   599.2  2384.9  604.412385.583
   612.3 2388.19   622.1 2388.71   641.8 2386.88   694.2 2390.18   700.8 2393.88
   730.2 2417.94   785.9  2445.9   851.4 2480.68   890.7 2499.84   972.6 2544.46
  1015.2 2561.56  1044.7 2575.72  1077.4 2589.12  1116.8 2601.15  1133.1 2604.79
#Mann= 3 ,-1 , 0
       0     .12       0   589.4    .045       0  604.41     .12       0
#XS Ineff= 2 , 0
          509.86 2391.32  662.65         2390.69
Permanent Ineff=
       F       F
Bank Sta=589.4,604.41
XS Rating Curve= 0 ,0
Exp/Cntr=0.3,0.1

Type RM Length L Ch R = 1 ,12421.1 ,399.2,381.7,364.9
XS GIS Cut Line= 3
     2148522.606      219829.166      2148177.33      220247.697
     2147842.376      220741.835
#Sta/Elev= 30
       0 2504.32    98.1 2481.47   153.6 2465.74   179.8 2464.69   359.5 2425.14
   418.4 2414.46     438 2409.12   460.9 2401.02   470.7 2399.31   493.5 2389.28
   532.8 2379.69   542.6 2378.92   549.1 2379.74     559 2382.15   575.4 2381.31
   627.8  2384.3   644.2 2392.68   663.9 2398.45   778.7 2414.45   788.6 2414.55
   801.7 2409.35   814.8  2408.9   844.3 2414.43   873.8 2416.02     923 2430.86
   965.7 2434.93  1001.8 2441.13  1037.9  2444.9  1113.3 2455.44  1139.5 2460.38
#Mann= 3 ,-1 , 0
       0     .12       0   532.8    .045       0   549.1     .12       0
Bank Sta=532.8,549.1
XS Rating Curve= 0 ,0
Exp/Cntr=0.3,0.1

Type RM Length L Ch R = 1 ,12039.4 ,317.3,318.3,317.1
XS GIS Cut Line= 3
     2147799.854      219629.769     2147858.882      220259.978
     2147808.534      220737.408
#Sta/Elev= 30
       0 2474.63     105 2456.12   167.3    2443   236.1 2424.63   252.5 2423.15
   298.4 2410.39   337.8 2401.16   360.8 2394.72   396.8 2381.72   413.2 2378.93
   439.5 2378.27  450.772372.907   459.2 2372.12  467.522372.894   478.8  2375.2
   511.6 2375.51     528 2378.46   590.3 2380.53   600.2 2382.74   626.4 2392.84
   639.5  2392.8   659.1 2397.69   688.5 2401.61   727.7 2404.04   802.8 2414.84
   861.6 2432.66   959.6  2455.9    1051 2462.91  1080.4  2466.9    1113 2469.36
#Mann= 3 ,-1 , 0
       0     .12       0  450.77    .045       0  467.52     .12       0
Bank Sta=450.77,467.52
XS Rating Curve= 0 ,0
Exp/Cntr=0.3,0.1

Type RM Length L Ch R = 1 ,11721.1 ,340.6,350,362.7
XS GIS Cut Line= 3
      2147509.79      219613.492     2147542.991      220180.676
       2147637.2      220714.517
#Sta/Elev= 30
       0 2430.97     111  2420.7   218.8 2415.55   287.3 2407.29   336.3 2396.44
   401.6 2372.26   466.9  2371.9   486.5 2370.75   499.6 2368.26     542 2370.36
  557.572366.156   571.4 2365.67   575.7 2366.12   587.8 2372.03   597.5 2371.74
   607.3 2373.65   620.4 2372.84   653.1  2380.7   679.2  2381.7   695.5 2385.25
   728.2 2397.74     738 2403.13   747.8 2404.79   757.6 2409.18   767.4 2411.49
   835.9 2438.01   881.6 2462.24   914.3 2476.91  1074.3 2519.78  1110.2 2526.78
#Mann= 3 ,-1 , 0
       0     .12       0  557.57    .045       0   575.7     .12       0
Bank Sta=557.57,575.7
XS Rating Curve= 0 ,0
Exp/Cntr=0.3,0.1

Type RM Length L Ch R = 1 ,11371.1 ,347.7,350,345.5
XS GIS Cut Line= 3
     2147408.555      219593.889     2147222.166      220106.455
     2147012.004      220614.047
#Sta/Elev= 30
       0 2430.05    32.7 2426.65      62 2427.47   140.4 2435.99     196 2425.12
   241.7 2413.04   284.1 2405.51   342.9 2391.08   411.5 2381.78   437.6 2370.18
   473.6 2366.34   529.1 2363.81   537.9 2360.96   545.4 2360.56   552.9 2360.86
     565 2364.04   587.9 2365.07   620.6  2362.2   663.1  2372.1   692.6 2382.83
   728.5 2400.56   741.6 2403.74   751.4 2409.96     843 2454.53   914.9 2481.54
   934.6 2486.96   977.1 2512.65   990.1 2518.28  1016.3 2522.52  1094.8 2529.66
#Mann= 3 ,-1 , 0
       0     .12       0   537.9    .045       0   552.9     .12       0
#XS Ineff= 2 , 0
                          588.88         2366.95
Permanent Ineff=
       F       F
Bank Sta=537.9,552.9
XS Rating Curve= 0 ,0
Exp/Cntr=0.3,0.1

Type RM Length L Ch R = 1 ,11021.1 ,354.8,350,348.8
XS GIS Cut Line= 3
     2147124.546       219507.55     2146893.554       219998.41
     2146773.249      220551.339
#Sta/Elev= 30
       0 2493.65    78.4 2467.53   189.6 2434.93   238.6 2418.74   254.9 2417.03
   307.2 2401.37   356.2 2390.22   405.2 2376.37   473.9 2360.04   496.7 2358.28
   522.9 2358.88     535 2355.16   545.8 2354.85     550 2355.17   565.4 2358.28
   601.4 2358.81   614.4 2355.71   624.3 2357.72   640.6 2357.85   653.7 2363.99
     693 2372.62   719.1 2383.71   764.9 2408.38   774.7  2411.2   791.1 2419.46
   876.1 2452.29     899 2459.41   915.4 2462.79     971 2470.46  1108.4 2482.79
#Mann= 3 ,-1 , 0
       0     .12       0     535    .045       0     550     .12       0
#XS Ineff= 2 , 0
          512.22 2360.56
Permanent Ineff=
       F       F
Bank Sta=535,550
XS Rating Curve= 0 ,0
Exp/Cntr=0.3,0.1

Type RM Length L Ch R = 1 ,10671.1 ,354.6,350,345.8
XS GIS Cut Line= 3
     2146673.987      219435.596     2146561.019      219966.904
     2146455.493      220522.229
#Sta/Elev= 30
       0 2510.27    58.9  2486.9   134.2 2454.16   147.2 2445.77   160.3 2443.34
   170.2 2436.36   189.8 2426.73   232.3 2411.25   281.4 2396.78   363.2 2368.35
   399.2 2359.58   441.8 2355.08   500.6 2354.33   523.6 2351.83  532.882347.685
   543.2 2347.01     549 2347.69   556.2 2349.57   579.1 2349.74   588.9 2352.26
   611.8 2349.91   624.9 2352.42   644.5 2351.92   670.6 2358.29   709.8 2374.59
     749 2386.98   837.2 2403.38   912.4 2411.43  1007.2 2413.95  1108.4 2423.96
#Mann= 3 ,-1 , 0
       0     .12       0  532.88    .045       0     549     .12       0
#XS Ineff= 2 , 0
                           596.9         2355.81
Permanent Ineff=
       F       F
Bank Sta=532.88,549
XS Rating Curve= 0 ,0
Exp/Cntr=0.3,0.1

Type RM Length L Ch R = 1 ,10321.1 ,289,291.5,293.4
XS GIS Cut Line= 3
     2146215.951      219394.757     2146215.951      219939.438
     2146213.748      220492.908
#Sta/Elev= 30
       0  2541.6    45.7  2515.6    65.2 2503.39   127.2 2468.82   146.8 2456.05
   159.8 2452.89   176.1 2441.92     225 2415.14   335.9 2362.42   407.7 2351.16
     437 2349.62   476.2 2349.28   495.8 2344.66   525.1 2345.38   534.9 2342.43
   541.4 2341.84   551.2 2342.42   597.1 2346.17   626.6 2346.77   767.4 2360.84
   780.5 2364.52   813.2 2379.02   888.6 2402.82   947.5 2425.59     977 2434.97
   993.4 2438.34  1016.3  2440.9  1065.4 2441.04  1085.1 2445.68  1098.2 2450.35
#Mann= 3 ,-1 , 0
       0     .12       0   534.9    .045       0   551.2     .12       0
Bank Sta=534.9,551.2
XS Rating Curve= 0 ,0
Exp/Cntr=0.3,0.1
